--- TmmyCrk.prj (project) ---

Proj Title=TmmyCrk
Current Plan=p01
Default Exp/Contr=0,0
English Units
Geom File=g01
Flow File=f01
Plan File=p01
BEGIN DESCRIPTION:
END DESCRIPTION:
DSS Export Rating Curves= 0
DSS Export Rating Curve Sorted= 0
DSS Export Volume Flow Curves= 0
DXF OffsetX= 0
DXF OffsetY= 0
DXF ScaleX= 0
DXF ScaleY= 0

--- TmmyCrk.p01 (plan) ---

Plan Title=Floodplain
Program Version=4.00
Geom File=g01
Flow File=f01
K Sum by GR=0
Std Step Tol=0.01
Critical Tol=0.01
Num of Std Step Trials=20
Max Error Tol=0.3
Flow Tol Ratio=0.001
Split Flow NTrial=30
Split Flow Tol=0.02
Split Flow Ratio=0.02
Log Output Level=0
Friction Slope Method=1
Unsteady Friction Slope Method=2
Unsteady Bridges Friction Slope Method=1
Global Log Level=0
CheckData=False
Run HTab=0
Run UNet=0
Run PostProcess=0
UNET Theta=0
UNET Theta Warmup=0
UNET ZTol=0
UNET ZSATol=0
UNET MxIter=0
UNET MaxInSteps=0
UNET DtIC=0
UNET DtMin=0
UNET MaxCRTS=0
UNET WFStab=0
UNET SFStab=0
UNET WFX=0
UNET SFX=0
UNET DSS MLevel=0
UNET DZMax Abort=0
UNET Convert EG Bridges=0
UNET Use Existing IB Tables=0
UNET Froude Limit=0
UNET Froude Power=0
Write IC File=0
Echo Input=False
Echo Output=False
Write Detailed=0

--- TmmyCrk.f01 (steady flow) ---

Flow Title=NFF Regression Equation
Program Version=4.00
Number of Profiles=1
Profile Names=P100yr
River Rch & RM=TmmyCrk,Main      ,49801.1
802.7889
River Rch & RM=TmmyCrk,Main      ,47388.3
888.6882
River Rch & RM=TmmyCrk,Main      ,42529.3
979.3314
River Rch & RM=TmmyCrk,Main      ,42348.7
1157.460
River Rch & RM=TmmyCrk,Main      ,39090.9
1217.335
River Rch & RM=TmmyCrk,Main      ,38773.2
1376.991
River Rch & RM=TmmyCrk,Main      ,36385.6
1474.687
River Rch & RM=TmmyCrk,Main      ,32795.4
1623.489
River Rch & RM=TmmyCrk,Main      ,30988.8
1785.245
River Rch & RM=TmmyCrk,Main      ,26785.5
1900.997
River Rch & RM=TmmyCrk,Main      ,26396.1
2267.950
River Rch & RM=TmmyCrk,Main      ,24842.4
2303.981
River Rch & RM=TmmyCrk,Main      ,22118.7
2536.437
River Rch & RM=TmmyCrk,Main      ,21765.2
2884.038
River Rch & RM=TmmyCrk,Main      ,14938.9
3052.838
River Rch & RM=TmmyCrk,Main      ,6831.1
3390.219
River Rch & RM=TmmyCrk,Main      ,6334.2
3882.676
River Rch & RM=TmmyCrk,Main      ,6198.6
5809.559
River Rch & RM=TmmyCrk,Main      ,242.7
5893.809
Boundary for River Rch & Prof#=TmmyCrk,Main      ,1
Up Type=0
Dn Type=3
Dn Slope=0.01023

--- TmmyCrk.g01 (geometry) ---

Geom Title=USGS 3m DEM
Program Version=4.10

River Reach=TmmyCrk         ,Main
Reach XY= 30
     1914286.082      216379.942     1911311.899      215984.231
     1910788.636      216490.646     1909958.894      216330.453
     1909444.606      216942.632     1907432.324      215270.642
      1905489.39      216107.991     1903903.725      214847.296
     1901083.889      214229.296     1899142.294      214666.108
     1896396.843      216981.423     1895221.844      217026.628
     1893382.211      216236.858     1892425.005      216325.821
     1891823.238      216816.911     1889358.781      216818.308
      1888552.55      218313.685     1886429.377      218509.153
     1886177.878      219993.965     1885464.172      221126.351
     1884375.314      220536.025     1883678.459      220911.192
     1881903.237      220566.886     1881324.753      221500.047
     1880311.362      221545.679     1878184.231      220429.475
     1877654.052      219591.951     1876918.121      219959.305
     1876289.142      219432.439     1875074.879      219646.089

Type RM Length L Ch R = 1 ,49801.1 ,198.3,213.3,227.9
XS GIS Cut Line= 3
     1914078.768      216155.557     1914170.342      216268.678
     1914644.907       216804.64
#Sta/Elev= 30
       0 2779.68    38.8 2765.04    87.3 2745.33      97 2743.58   116.4 2733.34
   165.4 2713.04   185.3 2705.93   205.2 2700.26     235 2693.65     245 2692.16
   264.8 2686.49   274.8 2685.36   284.7  2685.3   295.8  2685.3   310.8 2685.41
   324.5 2686.32   344.4 2689.49   394.1 2693.05   443.8 2700.88   473.6 2711.78
   483.6 2714.18   523.4 2732.18     593 2760.19   602.9 2761.25   622.8 2766.57
   722.2 2789.18   732.2 2790.92   821.6 2801.23   841.5 2803.14   861.4 2803.64
#Mann= 3 , 0 , 0
       0      .1       0   295.8    .045       0   310.8      .1       0
Bank Sta=295.8,310.8
XS Rating Curve= 0 ,0
Exp/Cntr=0.3,0.1

Type RM Length L Ch R = 1 ,49587.8 ,390.2,399.4,412.5
XS GIS Cut Line= 2
     1914098.968      216253.865     1914152.087       216978.75
#Sta/Elev= 30
       0 2748.17    19.9 2741.56    59.7 2724.43    69.7 2724.35   129.4 2701.12
   139.4 2697.61   159.3 2692.11   169.3 2691.97   199.1 2686.73   212.7 2683.86
     219 2682.76   227.7 2683.12   248.9 2686.08   258.9 2686.31   348.5 2696.66
   358.4 2696.96   368.4 2698.21   398.3 2704.71   438.1  2716.1     448 2716.99
     458 2719.06   527.7 2739.36   537.6 2740.52   557.6 2743.77   597.4 2747.21
   627.3 2750.45   647.2 2751.74     687 2755.45   716.9 2759.06   726.8 2759.77
#Mann= 3 , 0 , 0
       0      .1       0   212.7    .045       0   227.7      .1       0
Bank Sta=212.7,227.7
XS Rating Curve= 0 ,0
Exp/Cntr=0.3,0.1

Type RM Length L Ch R = 1 ,49188.3 ,292,300,297.7
XS GIS Cut Line= 3
     1913910.627      215875.942     1913726.757      216409.549
     1913465.783      216885.474
#Sta/Elev= 30
       0 2806.86      99 2799.17   207.9 2788.38   227.7 2784.65   257.4 2773.35
   277.2 2768.55   316.8 2749.93   356.5 2733.46   366.4 2732.72   455.5 2695.83
   475.3 2691.46     505 2679.71   556.9 2668.09   571.9 2666.93   574.3 2666.81
     594 2668.38   653.2 2679.58   682.8  2683.4   732.2 2695.61   771.6 2707.09
   791.4 2710.16     821 2721.87   860.5 2731.35   870.3 2732.62   890.1 2731.06
   978.9 2737.52  1018.4 2739.07  1038.1 2738.28  1087.4 2740.02  1107.2 2738.93
#Mann= 3 , 0 , 0
       0      .1       0   556.9    .045       0   571.9      .1       0
Bank Sta=556.9,571.9
XS Rating Curve= 0 ,0
Exp/Cntr=0.3,0.1

Type RM Length L Ch R = 1 ,48888.3 ,314.1,300,293.4
XS GIS Cut Line= 3
     1913823.287      215824.807     1913479.468      216243.752
     1913249.502      216765.843
#Sta/Elev= 30
       0 2785.06    19.7 2782.55    39.4 2777.48    88.7 2771.56   147.8 2759.06
   167.5 2751.32   206.9 2739.96   256.2 2727.82   275.9 2724.14   295.6 2718.11
   384.3 2697.79     404 2695.47   433.6 2686.57   502.6 2670.93   512.4  2669.9
   534.5 2660.75   549.5 2658.92     552  2658.9     602 2665.08     622 2666.37
   692.1 2676.61   712.1 2684.18   732.1 2690.06   812.2 2732.05   822.2 2734.28
   862.2 2749.62   882.3 2755.72   912.3 2759.78  1022.4 2769.25  1112.5 2771.56
#Mann= 3 , 0 , 0
       0      .1       0   534.5    .045       0   549.5      .1       0
Bank Sta=534.5,549.5
XS Rating Curve= 0 ,0
Exp/Cntr=0.3,0.1

Type RM Length L Ch R = 1 ,48588.3 ,309.8,310.7,310.4
XS GIS Cut Line= 3
     1913233.719      215611.291     1913217.088      216183.846
     1913172.665      216742.035
#Sta/Elev= 30
       0 2798.45    69.1  2795.6   118.5 2789.58   187.6 2789.45   197.5 2786.79
   217.3 2778.12     237 2773.73   306.2 2740.72   325.9 2736.19   404.9 2698.68
   414.8 2695.41   424.7 2694.08     474 2671.31   493.8 2666.17   513.5 2664.39
   565.3 2655.98   580.3 2654.97   582.8 2654.91   612.8 2656.55   652.8 2666.36
   692.8 2679.46   702.8 2679.54   782.8  2711.2   792.8 2711.25   882.8  2747.7
   892.8 2747.88   912.8 2754.73   972.8 2760.79  1012.8 2763.49  1132.8 2768.85
#Mann= 3 , 0 , 0
       0      .1       0   565.3    .045       0   580.3      .1       0
Bank Sta=565.3,580.3
XS Rating Curve= 0 ,0
Exp/Cntr=0.3,0.1

Type RM Length L Ch R = 1 ,48277.6 ,260.1,257.5,255
XS GIS Cut Line= 2
     1912961.027      215851.433     1912910.909      216704.228
#Sta/Elev= 30
       0 2752.68    69.5 2720.95    79.5 2720.03    89.4 2716.54   158.9 2688.16
   168.9 2687.06   178.8  2684.3   218.5 2668.16   238.4 2661.22   258.3  2655.9
   282.2 2652.49   288.1 2651.55   297.2 2651.61   377.5 2659.79   437.1  2669.2
   456.9 2671.17   476.8 2675.96   496.7 2682.57   536.4 2699.86   556.3 2704.45
   625.8  2737.4   635.7 2740.58   645.7 2741.74   655.6 2745.82   665.5  2748.3
   695.3 2750.44   764.9 2745.55   784.7 2745.05   834.4 2747.96   854.3 2751.04
#Mann= 3 , 0 , 0
       0      .1       0   282.2    .045       0   297.2      .1       0
Bank Sta=282.2,297.2
XS Rating Curve= 0 ,0
Exp/Cntr=0.3,0.1

Type RM Length L Ch R = 1 ,48020.1 ,260.9,269.4,277.9
XS GIS Cut Line= 3
     1912690.565      215629.311     1912691.692      216361.374
     1912695.283      216691.759
#Sta/Elev= 30
       0 2725.43    19.8 2722.56    39.6 2716.21    59.4 2708.05    79.1 2697.42
      89 2695.11   247.3  2704.5   267.1 2704.87   296.8  2702.1   346.2 2681.92
   375.9 2672.77     465 2657.38   546.9 2647.36   561.9 2646.21   563.9 2646.16
   583.7 2647.61   662.8 2666.51   672.7 2666.83   682.6 2669.39   712.3 2678.83
   751.5  2694.8   761.2 2695.86   800.1 2709.15   848.7 2711.92   926.4 2712.27
   945.8 2716.67   955.6 2717.11  1013.9 2733.88    1043 2740.56  1062.5 2742.54
#Mann= 3 , 0 , 0
       0      .1       0   546.9    .045       0   561.9      .1       0
Bank Sta=546.9,561.9
XS Rating Curve= 0 ,0
Exp/Cntr=0.3,0.1

Type RM Length L Ch R = 1 ,47750.5 ,365,362.3,358.3
XS GIS Cut Line= 3
     1912603.142      215714.916     1912377.635       216283.02
     1912275.251      216822.678
#Sta/Elev= 30
       0 2713.16     9.9 2710.47    19.7 2710.82    49.3 2699.12      69 2688.88
    88.7 2680.56    98.6 2676.96   108.4 2675.23     138 2673.43   177.4 2672.67
   226.7 2669.03   285.9 2663.49   384.5 2652.09   483.1 2644.41   492.9 2643.88
   502.8 2644.01   611.2 2650.51   741.1 2655.82     801 2663.73     821 2665.35
   890.9 2674.84   910.8  2676.1   970.8 2683.52  1000.7 2688.84  1010.7 2688.94
  1030.7 2693.07  1060.6  2700.9  1090.6 2705.87  1100.6 2705.63  1160.5 2711.93
#Mann= 3 , 0 , 0
       0      .1       0   483.1    .045       0   502.8      .1       0
Bank Sta=483.1,502.8
XS Rating Curve= 0 ,0
Exp/Cntr=0.3,0.1

Type RM Length L Ch R = 1 ,47388.3 ,308,298.8,290.4
XS GIS Cut Line= 3
     1912249.704       215489.97     1912111.424      216018.578
     1912002.465      216565.901
#Sta/Elev= 30
       0 2786.76    59.6 2784.17   129.2 2769.03   139.1 2767.39     149 2767.37
   218.6 2754.12   238.4 2743.65   248.4 2742.59   258.3 2739.13     308 2717.13
   327.8 2709.58   347.7 2706.02   427.2 2676.46   437.1 2676.43   476.8  2660.6
   526.5 2647.53   546.4 2644.22   556.4 2643.09   566.3  2644.5   616.2 2659.95
   636.1  2663.7     666 2674.63   715.8 2691.04   725.8 2691.66   765.6 2703.81
   815.5 2717.08   855.3 2720.18   925.1 2720.77   974.9  2722.7  1104.5 2730.39
#Mann= 3 , 0 , 0
       0     .06       0   546.4    .045       0   566.3     .06       0
Bank Sta=546.4,566.3
XS Rating Curve= 0 ,0
Exp/Cntr=0.3,0.1

Type RM Length L Ch R = 1 ,47089.2 ,304,309.9,315.8
XS GIS Cut Line= 3
     1911744.192      215472.701     1911822.584      216010.144
     1911916.634      216564.484
#Sta/Elev= 30
       0 2777.29    49.4 2773.34   167.9 2766.76   197.5 2761.25     237 2750.92
   256.8 2748.14   296.2 2735.92   335.8 2720.97   345.6 2720.03   434.5  2679.4
   444.4 2679.23   503.6 2653.26   523.4 2643.71   535.6 2642.02   550.6 2640.51
     553 2640.47   592.4 2649.24     622 2658.45   641.8 2661.85   710.8 2685.29
   720.7 2688.14   730.6 2689.01   799.6 2712.33   819.3  2716.8   829.2 2717.03
   868.6 2722.45   908.1 2726.24   927.8 2727.16   996.9 2734.71  1105.4 2743.32
#Mann= 3 , 0 , 0
       0     .06       0   535.6    .045       0   550.6     .06       0
Bank Sta=535.6,550.6
XS Rating Curve= 0 ,0
Exp/Cntr=0.3,0.1

Type RM Length L Ch R = 1 ,46779.2 ,342.4,325.1,305.4
XS GIS Cut Line= 3
      1911595.48      215496.411     1911517.391      216217.729
     1911635.959      216615.284
#Sta/Elev= 30
       0 2761.56    89.4 2745.86   188.8 2732.12   218.6 2724.28   228.6 2724.05
   248.5 2719.71   278.3 2711.17   308.1 2700.72     318 2700.57   367.7 2681.77
   387.6 2675.87   417.4  2670.3   496.9 2647.34   516.8  2644.1   535.3  2636.9
   546.6 2635.49   550.3 2635.87   606.3 2642.95   616.2 2645.42   675.8 2668.51
   695.7 2673.42   774.9 2701.58   784.8 2704.37   794.7 2704.36   834.2 2716.63
   853.9 2721.37   873.7 2722.94   923.1 2723.24    1012  2729.4  1140.4 2731.51
#Mann= 3 , 0 , 0
       0     .06       0   535.3    .045       0   550.3     .06       0
Bank Sta=535.3,550.3
XS Rating Curve= 0 ,0
Exp/Cntr=0.3,0.1

Type RM Length L Ch R = 1 ,46454.1 ,223.6,223.2,221.6
XS GIS Cut Line= 3
     1911000.893      215533.681     1911184.313       215927.52
     1911541.182      216450.031
#Sta/Elev= 30
       0 2758.33      79 2763.58    98.7 2764.08   108.6 2762.32   148.1 2742.68
   177.7 2731.86   187.6 2729.28   197.5 2728.38   246.8  2714.7   286.4 2699.95
   296.2 2698.66     395 2674.26   434.5 2666.32   454.2  2657.8   493.8 2645.26
   513.6 2641.22   553.1 2629.33   565.7 2627.66   572.9 2627.62   580.7 2628.04
   612.4 2631.15   642.1 2636.78   731.1  2669.3   740.9 2670.45   780.5 2685.67
   849.7 2707.95   869.5 2710.25   899.1 2716.89   958.4 2725.27  1067.2 2726.12
#Mann= 3 , 0 , 0
       0     .06       0   565.7    .045       0   580.7     .06       0
Bank Sta=565.7,580.7
XS Rating Curve= 0 ,0
Exp/Cntr=0.3,0.1

Type RM Length L Ch R = 1 ,46229.6 ,294.3,300.5,308.9
XS GIS Cut Line= 3
     1910768.841      215747.613     1911138.871      216222.936
     1911510.549      216661.614
#Sta/Elev= 30
       0 2749.96    69.1 2750.97   246.9 2745.91   256.8 2743.43   286.4 2732.47
   296.2  2727.7     316 2721.58   404.9 2687.45   424.6 2682.07   434.5 2676.78
     474 2659.93   523.4 2641.24   533.2 2638.04     553 2634.53   572.8 2628.16
   594.9 2625.45   609.9 2625.05   612.3 2625.04   632.1 2627.64   691.6 2642.92
   711.4 2651.63   800.6 2681.58   830.4 2695.61   850.2 2699.81   879.9  2703.7
   919.6 2706.88   939.4 2707.12   959.2 2709.72  1048.5 2716.79  1177.3 2720.46
#Mann= 3 , 0 , 0
       0     .06       0   594.9    .045       0   609.9     .06       0
Bank Sta=594.9,609.9
XS Rating Curve= 0 ,0
Exp/Cntr=0.3,0.1

Type RM Length L Ch R = 1 ,45929.6 ,293.3,299.9,307.8
XS GIS Cut Line= 3
     1910706.087       215787.96     1910939.018      216392.686
     1911112.573      216913.833
#Sta/Elev= 30
       0 2746.13    49.8 2744.12   189.4 2734.54   229.3 2733.42   289.1 2734.35
     319 2731.63   398.8 2698.03   418.7 2692.86   508.5 2646.88   518.4 2646.37
   548.3 2635.15   578.2 2626.64   598.2 2622.65   618.1 2621.09   640.5 2617.51
   655.5 2617.11     658  2617.1     668 2618.17     688 2623.73   727.9 2630.99
   807.8 2658.91   817.8 2659.37   857.8 2673.34   877.7 2678.51   957.6 2683.63
  1007.6 2690.16  1017.6 2690.39  1127.4 2705.28  1167.4 2708.42  1197.3 2713.15
#Mann= 3 , 0 , 0
       0     .06       0   640.5    .045       0   655.5     .06       0
Bank Sta=640.5,655.5
XS Rating Curve= 0 ,0
Exp/Cntr=0.3,0.1

Type RM Length L Ch R = 1 ,45629.6 ,315.1,321.3,325.1
XS GIS Cut Line= 3
     1910630.605      215807.235     1910675.097      216494.808
     1910651.991      217015.058
#Sta/Elev= 30
       0 2740.84    89.9 2733.43   199.7 2721.34   229.7 2716.89   259.6 2709.97
   279.6  2708.1   349.5 2695.99   369.5  2694.2   449.4 2676.17   459.3 2675.38
   469.3  2671.5   509.3 2652.02   539.2 2642.73   559.2 2640.13   629.1 2626.02
   649.1 2624.24   681.5 2617.05   696.5 2614.59   698.8 2614.42   708.7 2615.95
   738.1 2624.31     748 2624.38   826.6 2651.82   836.4 2652.22     915 2673.46
   934.6 2675.52     974 2683.81  1121.3 2692.37    1200 2710.84  1209.8 2711.13
#Mann= 3 , 0 , 0
       0     .06       0   681.5    .045       0   696.5     .06       0
Bank Sta=681.5,696.5
XS Rating Curve= 0 ,0
Exp/Cntr=0.3,0.1

Type RM Length L Ch R = 1 ,45308.1 ,284.8,275.3,266.2
XS GIS Cut Line= 3
     1910569.358      215799.905     1910402.838      216540.616
     1910382.793      216976.343
#Sta/Elev= 30
       0 2735.55    79.9 2726.44    99.9 2725.34   199.8 2715.48   249.7 2709.16
   269.7 2703.48   279.7  2703.3   339.6 2680.38   369.6 2667.07   379.6 2665.66
   389.6 2662.28   459.5 2628.81   479.5 2623.86     518 2605.98   529.4 2604.79
     533 2605.44   549.4 2608.78   569.4 2610.57   619.4  2618.8   659.3  2631.8
   669.3 2632.26   749.2 2660.98   759.2 2662.22   788.9 2670.34   798.8 2671.79
   937.6  2680.4  1076.4  2686.7  1106.2 2689.12  1145.8 2688.27  1195.4 2684.64
#Mann= 3 , 0 , 0
       0      .1       0     518    .045       0     533      .1       0
Bank Sta=518,533
XS Rating Curve= 0 ,0
Exp/Cntr=0.3,0.1

Type RM Length L Ch R = 1 ,45032.8 ,304.8,292,278.8
XS GIS Cut Line= 3
     1910090.174      215791.514     1910188.341      216305.085
     1910302.951      216975.017
#Sta/Elev= 30
       0 2696.25    78.9 2708.56   118.4 2710.65   138.1 2709.41   167.7 2704.26
   187.4 2702.41   207.2    2699   246.6 2688.06   276.2 2677.73   286.1 2677.36
     365 2648.22   384.8 2644.45   453.8 2619.64   473.5 2616.35   522.9 2599.88
   532.9 2598.15   542.9 2600.24   562.8 2610.73   572.8 2611.28   652.8 2640.74
   662.8 2640.97   732.8 2664.86   742.8 2667.59   752.8 2668.89   802.7 2670.32
   912.7 2670.84  1132.6 2682.14  1142.6 2681.84  1182.5 2672.45  1202.5  2669.8
#Mann= 3 , 0 , 0
       0      .1       0   522.9    .045       0   542.9      .1       0
Bank Sta=522.9,542.9
XS Rating Curve= 0 ,0
Exp/Cntr=0.3,0.1

Type RM Length L Ch R = 1 ,44740.7 ,301.7,308,308
XS GIS Cut Line= 3
     1909558.328      215982.183     1909991.551      216453.042
       1910226.8      216995.625
#Sta/Elev= 30
       0 2678.07     110 2696.67     130 2702.14     180 2711.34     190 2712.25
     200  2711.7   239.9 2707.88   259.9  2703.2   269.9 2698.97   469.9  2605.6
   489.9 2598.14   499.9 2591.31   509.9  2588.7   519.9 2588.77   599.8 2599.68
   619.8 2603.47   639.8 2605.61     699 2611.72   728.5 2611.58     768 2614.39
   797.5 2617.64   827.1 2622.56   856.7 2630.86   965.1 2653.49    1044 2662.78
  1132.7 2675.49  1152.4 2676.97  1162.2  2676.5  1211.5 2669.24  1231.2 2665.32
#Mann= 3 , 0 , 0
       0      .1       0   509.9    .045       0   519.9      .1       0
Bank Sta=509.9,519.9
XS Rating Curve= 0 ,0
Exp/Cntr=0.3,0.1

Type RM Length L Ch R = 1 ,44432.8 ,293.6,299.7,304.5
XS GIS Cut Line= 3
      1909501.79       216021.06     1909820.332      216652.791
     1910169.387      217035.122
#Sta/Elev= 30
       0 2666.55    49.8 2671.15    89.7 2677.24   209.3 2703.29   318.9 2698.23
   328.8 2696.72   368.7 2684.48   448.4 2654.97   468.3  2650.1   488.3 2643.03
   518.2 2630.04   587.9 2617.23   617.8 2609.89   677.6  2589.1   687.6 2582.75
   697.5 2579.14     700 2579.42     715 2582.41   737.4 2588.97     817 2605.43
   836.9 2611.78   906.6 2629.04   926.5 2632.05   996.2 2651.25  1065.9 2660.65
  1095.8 2666.23  1115.7 2667.56  1185.4 2660.56  1205.3 2660.03  1225.2 2657.17
#Mann= 3 , 0 , 0
       0      .1       0     700    .045       0     715      .1       0
Bank Sta=700,715
XS Rating Curve= 0 ,0
Exp/Cntr=0.3,0.1

Type RM Length L Ch R = 1 ,44132.8 ,191.9,208.3,232.2
XS GIS Cut Line= 3
     1909439.679        216061.4     1909601.316      216853.115
     1909860.212      217281.627
#Sta/Elev= 30
       0 2658.42    39.9 2662.67    79.8 2670.36   159.6 2680.57   219.5 2681.85
   289.3 2675.78   369.1 2652.24   379.1  2652.6   458.9 2629.65   558.6 2616.07
   628.5 2612.54   678.4 2612.98   698.3  2606.3   758.2 2580.76   768.1 2580.36
   788.1 2571.85   798.1 2571.06   800.5 2571.17   815.5 2572.32   925.8 2578.37
   974.9 2585.89   984.8 2585.65    1024 2596.65  1073.1 2606.32  1092.7 2607.21
  1161.4 2629.62  1190.9  2636.2  1210.5 2636.86  1279.2 2649.74  1308.7 2649.66
#Mann= 3 , 0 , 0
       0     .06       0   800.5    .045       0   815.5     .06       0
Bank Sta=800.5,815.5
XS Rating Curve= 0 ,0
Exp/Cntr=0.3,0.1

Type RM Length L Ch R = 1 ,43924.7 ,111.6,126.6,141.5
XS GIS Cut Line= 3
     1909550.795      216732.833     1909479.421      216837.873
      1909297.62      217152.995
#Sta/Elev= 30
       0  2604.2    19.5 2600.74    48.8 2594.65    68.4  2590.1    87.9  2584.1
    97.7 2582.43   107.5 2576.07   117.2  2571.2     127 2570.23   205.7 2567.92
   215.5 2567.45   231.8 2565.97   235.2 2565.65     245 2565.99   246.8 2566.38
   254.8 2568.11   264.6 2573.17   274.5 2579.26   294.2 2589.89     304 2591.63
   313.8 2595.74   333.5  2606.8   353.1  2616.8   372.8 2624.54   392.5 2630.82
   402.3 2633.12   412.1 2634.14   431.8 2639.82   461.3 2645.82   490.8 2652.55
#Mann= 3 , 0 , 0
       0     .06       0   231.8    .045       0   246.8     .06       0
Bank Sta=231.8,246.8
XS Rating Curve= 0 ,0
Exp/Cntr=0.3,0.1

Type RM Length L Ch R = 1 ,43798.1 ,295.7,279.6,263.4
XS GIS Cut Line= 3
     1909379.443      216067.845     1909464.608       216790.74
     1908962.298      216991.394
#Sta/Elev= 30
       0 2654.31    89.7 2661.43   169.5 2670.17   229.3 2672.08   239.3  2670.8
   259.2 2664.61   269.2 2663.96     359 2627.82   368.9 2627.66   408.8 2613.49
   448.7 2602.73   458.7 2603.01   548.4 2585.94   638.2 2575.65   727.9  2571.2
     845 2562.11   855.7 2561.75     860 2562.21   865.6 2562.81   944.3 2600.17
   963.9 2611.59   983.6 2609.89  1032.8 2598.19  1052.4 2591.03  1081.9 2585.14
  1121.3 2594.02    1141 2602.38  1209.8 2619.08  1229.5 2626.15  1268.8 2634.56
#Mann= 3 , 0 , 0
       0     .06       0     845    .045       0     860     .06       0
Bank Sta=845,860
XS Rating Curve= 0 ,0
Exp/Cntr=0.3,0.1

Type RM Length L Ch R = 1 ,43518.5 ,274.3,271.6,272.2
XS GIS Cut Line= 3
     1909364.158      216043.607     1909320.513      216538.911
     1909137.366      216897.127
#Sta/Elev= 30
       0 2651.77     9.9 2651.78    99.4 2659.01   109.4    2659   188.9 2664.94
   248.6 2666.75   258.6 2664.36   278.4 2656.03   288.4 2654.99   298.3 2651.72
   377.9 2616.49   387.8 2614.98   397.8 2612.04   437.6 2594.48   467.4 2582.39
   487.3 2578.13   526.7 2560.74   536.7 2558.07   546.3 2557.98   551.7 2558.53
   585.5 2561.64   634.6 2567.58   683.7 2579.88   693.5 2579.28   713.1 2582.28
   742.5 2582.98   791.6  2580.3   830.8 2581.11   840.7 2579.76   899.5 2583.92
#Mann= 3 , 0 , 0
       0      .1       0   536.7    .045       0   551.7      .1       0
Bank Sta=536.7,551.7
XS Rating Curve= 0 ,0
Exp/Cntr=0.3,0.1

Type RM Length L Ch R = 1 ,43246.9 ,294.5,300,304.3
XS GIS Cut Line= 3
     1909231.933       215998.22     1909035.957      216532.504
     1908777.555      217009.279
#Sta/Elev= 30
       0 2634.46    49.9 2640.65    59.9 2640.54    89.9 2645.99   109.8 2648.03
   239.6 2653.92   279.6 2653.57   339.5  2629.9   359.4 2626.02   439.3 2596.41
   459.3 2591.37   549.1 2558.83   561.6 2557.85   569.1 2556.03     579 2555.97
   588.8  2559.4   608.5 2569.93     648 2587.12   667.7 2592.32   746.6 2625.09
   766.3 2629.44   795.9 2640.71   825.4 2643.76   884.6 2646.32   914.2 2649.05
   963.5 2657.71  1042.4 2668.72    1072 2677.09  1081.8 2677.78  1111.4 2686.68
#Mann= 3 , 0 , 0
       0      .1       0   561.6    .045       0     579      .1       0
Bank Sta=561.6,579
XS Rating Curve= 0 ,0
Exp/Cntr=0.3,0.1

Type RM Length L Ch R = 1 ,42946.9 ,420.7,417.5,412.1
XS GIS Cut Line= 3
     1909090.859      215922.378     1908776.996       216388.99
     1908432.586      216808.654
#Sta/Elev= 30
       0 2601.93    19.7 2603.63    49.3 2603.65     148 2615.37   157.8 2614.96
   246.6 2621.75   266.4 2621.14   315.7 2624.89   325.6 2624.28   345.3 2619.96
     365 2614.04   374.9 2612.46   434.1 2582.18   473.6 2566.78   554.8  2554.6
   562.4 2554.12   569.8  2555.4   582.1  2560.1     592 2565.34   680.8 2592.94
   720.3 2602.35     740 2609.81     819 2622.78   848.6 2628.88   868.4 2635.19
   917.7 2640.07   976.9    2641  1006.5 2647.41  1075.6 2658.51  1105.2 2665.42
#Mann= 3 , 0 , 0
       0      .1       0   554.8    .045       0   569.8      .1       0
Bank Sta=554.8,569.8
XS Rating Curve= 0 ,0
Exp/Cntr=0.3,0.1

Type RM Length L Ch R = 1 ,42529.3 ,178,180.5,181.2
XS GIS Cut Line= 2
     1908641.639      215782.154     1908229.743       216610.18
#Sta/Elev= 30
       0 2646.59    79.6  2645.3    99.4 2642.01   129.3 2632.33     169 2615.17
     179    2614   218.8 2597.76   268.5 2580.13   278.4 2576.88   298.3 2573.37
     348 2557.25     358 2552.96   370.7 2550.97   377.9  2550.8   385.7  2550.8
   397.8 2551.16   417.7 2555.62   447.5 2559.24   497.2 2572.43   517.1 2579.62
   586.7 2600.34   606.6 2603.95   686.2 2623.78     706 2626.42   795.5 2643.98
   805.5 2644.49   845.3  2658.4     895 2684.13   904.9  2684.6   924.8 2694.37
#Mann= 3 , 0 , 0
       0      .1       0   370.7    .045       0   385.7      .1       0
Bank Sta=370.7,385.7
XS Rating Curve= 0 ,0
Exp/Cntr=0.3,0.1

Type RM Length L Ch R = 1 ,42348.7 ,297,292.8,290.4
XS GIS Cut Line= 3
      1908621.03      215562.973     1908323.409      216020.062
     1908062.134      216503.079
#Sta/Elev= 30
       0 2624.78     9.9 2623.71    79.3  2629.5   109.1 2630.77     119 2629.94
   208.3 2638.51   267.8  2637.8     357 2618.96   376.8 2612.42   396.7 2603.44
   436.4 2588.28   456.2 2583.96   545.4 2551.38   552.9 2550.96   565.4 2550.79
   575.4  2551.1   585.4  2553.2   625.3 2571.47   655.3 2582.61   665.3 2585.26
   675.2  2585.7   765.1 2607.22   775.1 2606.48     805 2612.26     835 2615.23
   884.9 2615.12   984.8 2621.12  1054.7 2631.66  1084.6 2639.04  1094.6 2638.31
#Mann= 3 , 0 , 0
       0      .1       0   552.9    .045       0   575.4      .1       0
Bank Sta=552.9,575.4
XS Rating Curve= 0 ,0
Exp/Cntr=0.3,0.1

Type RM Length L Ch R = 1 ,42056   ,308.7,324.1,339.5
XS GIS Cut Line= 3
     1908371.585      215440.824     1908095.946      215812.273
     1907845.745      216422.077
#Sta/Elev= 30
       0 2657.87    29.5 2651.14    39.4 2651.36    98.4 2635.72   137.8 2622.85
   157.5 2620.46   206.7 2605.96   255.9 2594.84   265.7 2593.43   275.6 2593.96
   354.3 2573.85   364.1 2572.34   403.5 2569.94   462.6 2568.88   574.2 2547.39
   589.2 2547.15   592.4 2547.14   612.4 2553.08   692.2  2580.8   702.2 2581.98
   782.1 2610.65   802.1 2614.12     882 2635.82     902 2639.32   971.9 2657.02
   991.9 2664.71  1001.8 2666.06  1091.7 2698.71  1101.7 2700.66  1121.7 2708.71
#Mann= 3 , 0 , 0
       0      .1       0   574.2    .045       0   589.2      .1       0
Bank Sta=574.2,589.2
XS Rating Curve= 0 ,0
Exp/Cntr=0.3,0.1

Type RM Length L Ch R = 1 ,41731.8 ,290.2,273.2,256.2
XS GIS Cut Line= 3
     1908246.614      215466.134     1907675.624      215776.768
     1907512.466      216178.403
#Sta/Elev= 30
       0  2655.4      90 2637.54     110 2631.15     180 2616.61     270 2590.59
     290 2582.16     310 2576.65     360 2565.68     430 2547.16     440  2545.8
     450 2545.69     460 2546.83     470 2553.73     480 2556.71     550 2572.26
     560 2576.38     580  2580.5     600 2586.38     640  2599.6     650 2604.79
   699.3 2624.53   709.1 2625.49   748.5 2639.67     788 2649.74   837.2 2657.34
   906.2 2681.08     916 2681.45   935.7 2686.16   994.9 2694.36  1083.5 2701.77
#Mann= 3 , 0 , 0
       0      .1       0     440    .045       0     460      .1       0
Bank Sta=440,460
XS Rating Curve= 0 ,0
Exp/Cntr=0.3,0.1

Type RM Length L Ch R = 1 ,41458.5 ,277.1,278.9,280.7
XS GIS Cut Line= 3
     1908051.415      215116.606     1907718.732      215329.501
     1907450.293      216129.865
#Sta/Elev= 30
       0 2650.34    49.4 2635.54    69.1  2634.1    88.9 2640.67   138.2 2652.46
   167.9 2657.06   177.7 2655.67   246.9 2635.14   266.6 2627.32   345.6 2603.63
   365.4  2595.5   414.8 2581.08   434.7 2577.96   524.1 2555.42     534 2554.87
   571.3 2546.05   583.7 2545.71   586.3 2545.94   633.3 2555.14   712.8 2580.74
   732.6  2584.4   812.1  2612.7     822 2615.87     832 2616.82   881.6 2635.03
   891.6 2637.37  1010.7 2655.69  1020.7 2655.76    1110 2678.29  1239.2 2688.89
#Mann= 3 , 0 , 0
       0      .1       0   571.3    .045       0   586.3      .1       0
Bank Sta=571.3,586.3
XS Rating Curve= 0 ,0
Exp/Cntr=0.3,0.1

Type RM Length L Ch R = 1 ,41179.3 ,324.1,304.3,284.5
XS GIS Cut Line= 3
     1907694.949      214815.218     1907417.062      215464.339
     1907401.801      216094.982
#Sta/Elev= 30
       0  2635.6    39.8 2631.03    59.7 2632.22   149.2  2631.5   218.8 2624.78
   278.5 2615.03   318.2 2599.11     358    2588   377.9 2584.07   387.9 2583.45
   457.5 2562.84   487.3 2551.22   497.2 2550.51   507.2 2546.44   516.6 2544.37
   517.1 2544.26   531.6 2544.84   596.7 2551.59   616.6 2555.77   666.3 2569.83
   686.2 2577.25   696.2 2579.26     785 2609.76   794.8  2609.9   863.8  2621.2
   972.2  2627.2  1129.9  2644.1  1267.9 2654.99  1297.5 2659.43  1336.9 2667.71
#Mann= 3 , 0 , 0
       0      .1       0   516.6    .045       0   531.6      .1       0
Bank Sta=516.6,531.6
XS Rating Curve= 0 ,0
Exp/Cntr=0.3,0.1

Type RM Length L Ch R = 1 ,40875   ,249.5,240.1,230.8
XS GIS Cut Line= 3
     1906982.103      214894.762      1907268.56      215463.001
     1907330.685      216107.026
#Sta/Elev= 30
       0 2618.79    19.9 2626.04    29.8  2627.8     169 2636.31   208.8 2636.73
   238.6  2634.8   248.6 2632.17   278.4  2619.5   298.3 2618.13   397.7 2578.76
   417.6 2574.61   487.2 2544.27   498.6 2540.59   507.1 2539.71   513.6  2540.1
     527 2542.73   546.9 2549.78   616.5  2569.8   626.4 2570.38     706 2596.53
     716 2596.75   775.7 2611.22   805.6 2614.95   875.3 2619.81   974.8  2619.1
  1094.2 2621.24  1134.1 2627.52  1193.8 2629.32  1243.6 2636.95  1283.4 2645.92
#Mann= 3 , 0 , 0
       0      .1       0   498.6    .045       0   513.6      .1       0
Bank Sta=498.6,513.6
XS Rating Curve= 0 ,0
Exp/Cntr=0.3,0.1

Type RM Length L Ch R = 1 ,40634.9 ,343.3,363.7,384.2
XS GIS Cut Line= 3
     1906617.605      215159.154     1907133.508      215584.082
     1907266.049      216143.628
#Sta/Elev= 30
       0 2590.21    69.8 2612.74    89.8 2620.55    99.8 2622.06   279.3 2628.91
   289.3 2627.45   349.2 2612.43   379.1 2603.83     399 2595.07     409 2588.39
     429 2578.22   448.9 2575.44   508.8 2543.33   518.7 2538.44   521.5 2538.16
   528.7 2537.44   536.5  2538.8   568.6 2545.22   608.5 2551.31   618.5 2553.67
   628.5 2558.13   668.4 2567.96   757.6  2574.9   916.2 2583.01   965.8 2581.44
  1015.4 2586.53  1064.9    2599  1114.5 2605.17  1213.7 2620.92  1243.4 2628.07
#Mann= 3 , 0 , 0
       0      .1       0   521.5    .045       0   536.5      .1       0
Bank Sta=521.5,536.5
XS Rating Curve= 0 ,0
Exp/Cntr=0.3,0.1

Type RM Length L Ch R = 1 ,40270.4 ,296.4,292,284.7
XS GIS Cut Line= 3
     1906555.379      215194.287     1906852.538      215594.948
     1906831.322      216271.503
#Sta/Elev= 30
       0 2586.57    59.9  2608.7    69.8 2610.83    99.8 2621.18   249.4 2630.84
   309.3 2630.71   349.2 2622.59     409 2603.07     419 2602.12     429 2599.31
   518.7 2570.26   538.6 2566.79   598.4 2540.26   608.3 2537.28   628.2 2535.74
   638.2 2535.23   643.2 2535.73   658.1 2538.96   717.8 2557.13   727.8 2557.45
   807.4 2584.29   817.4 2584.42     897 2611.59     907 2611.58   936.8 2615.39
  1006.5 2616.81  1026.4 2619.11  1086.1 2633.65  1096.1 2634.05  1175.7  2661.6
#Mann= 3 , 0 , 0
       0      .1       0   628.2    .045       0   643.2      .1       0
Bank Sta=628.2,643.2
XS Rating Curve= 0 ,0
Exp/Cntr=0.3,0.1

Type RM Length L Ch R = 1 ,39978.1 ,300.7,300,303.9
XS GIS Cut Line= 3
     1906476.824      215213.086     1906575.042      215777.067
     1906732.482      216296.078
#Sta/Elev= 30
       0 2572.02    29.6 2580.91    39.5 2581.29   118.4 2604.59   138.2 2607.82
   167.8 2616.35   187.5  2618.7   296.1 2623.29   315.8  2617.6   325.7 2616.81
   404.7 2580.36   414.6 2580.02   503.4 2545.31   523.1  2542.3     565 2531.41
   582.3 2528.55   592.2 2528.96   611.9 2532.11   641.5 2548.89   700.7 2570.63
   720.4 2573.92   789.4 2598.47   799.3  2601.4   809.1 2601.41   848.6 2615.18
   927.5  2625.6   996.5 2640.35  1006.4 2640.37  1085.2 2662.73  1114.8  2667.9
#Mann= 3 , 0 , 0
       0      .1       0     565    .045       0   592.2      .1       0
Bank Sta=565,592.2
XS Rating Curve= 0 ,0
Exp/Cntr=0.3,0.1

Type RM Length L Ch R = 1 ,39678.1 ,308.5,303.1,296.1
XS GIS Cut Line= 3
     1906171.844      215232.258     1906282.968      215763.107
     1906356.406      216324.982
#Sta/Elev= 30
       0  2575.8     9.9 2575.41    88.8 2549.43   147.9 2536.82   157.8 2537.58
   187.4 2546.58   207.1 2549.72   246.5 2559.66   276.1 2565.13   345.1 2569.84
   364.9 2569.84   443.8 2554.95   473.3 2543.85   483.2 2540.92     493 2540.11
   534.9  2523.5   542.4 2521.33   549.9 2521.08   552.3    2521   582.1 2525.69
   631.8 2527.03   671.6 2538.02   681.5 2538.65   761.1 2566.44     781 2570.04
   860.5 2598.02   880.4 2600.92   930.1 2613.26  1029.5 2617.87    1109 2604.65
#Mann= 3 , 0 , 0
       0      .1       0   534.9    .045       0   549.9     .06       0
Bank Sta=534.9,549.9
XS Rating Curve= 0 ,0
Exp/Cntr=0.3,0.1

Type RM Length L Ch R = 1 ,39374.9 ,290.5,283.9,277.4
XS GIS Cut Line= 3
     1905836.445      215350.183     1906007.417      215877.849
     1906244.285      216368.095
#Sta/Elev= 30
       0 2615.47    59.4 2587.68    79.2 2584.05   138.7 2563.42   168.4 2555.51
   188.2 2553.28   257.5 2536.42   277.3 2533.86   326.9 2520.85   366.5 2515.92
   445.7 2510.59   534.9 2514.34   571.8 2510.97   584.4 2509.97   586.8 2510.06
   604.2 2512.49   643.8 2523.38   673.5 2538.57   683.4 2540.14   732.9 2565.17
   752.7 2572.23   762.6 2573.94     921 2595.23   960.6 2594.86   980.4 2591.54
  1000.2  2590.4  1029.8 2584.83  1059.5 2582.28  1069.4 2583.47  1099.1 2591.23
#Mann= 3 , 0 , 0
       0      .1       0   571.8    .045       0   586.8      .1       0
#XS Ineff= 2 , 0
          533.48  2514.4
Permanent Ineff=
       F       F
Bank Sta=571.8,586.8
XS Rating Curve= 0 ,0
Exp/Cntr=0.3,0.1

Type RM Length L Ch R = 1 ,39090.9 ,146,158.5,171
XS GIS Cut Line= 3
     1905762.818      215380.084     1905705.374      215958.191
      1906119.22      216423.871
#Sta/Elev= 30
       0 2605.13    29.5 2594.11    49.2 2590.73    78.8 2577.53    98.5 2571.41
   118.2 2567.12   137.8 2565.32   216.6 2549.03   236.3 2546.88   315.1 2527.97
   324.9 2527.86   344.6 2523.92   413.6 2520.77   482.5 2523.03   521.9 2522.61
   600.7 2507.35   640.3 2501.15     670 2493.76   679.8 2493.22   680.7 2493.31
   695.7 2495.08   828.2 2511.09   867.7 2517.62     937 2531.44   986.4 2544.23
  1055.6 2555.02    1115 2567.88  1144.6 2572.04  1184.2 2580.76    1204 2587.26
#Mann= 3 , 0 , 0
       0      .1       0   680.7    .045       0   695.7      .1       0
Bank Sta=680.7,695.7
XS Rating Curve= 0 ,0
Exp/Cntr=0.3,0.1

Type RM Length L Ch R = 1 ,38932.4 ,131.8,158.9,184.8
XS GIS Cut Line= 3
     1905689.561      215382.609     1905616.451      215981.985
     1905688.495      216394.266
#Sta/Elev= 30
       0 2616.83    29.7 2606.58    39.6 2606.63    49.5 2603.08    89.1 2582.12
   118.8 2572.75   128.7 2572.33   217.8 2556.14   306.9 2547.12   445.4 2550.43
   455.3 2548.04   465.2 2543.59   504.8  2522.2   514.7 2521.77   524.6 2518.31
   554.3 2511.98   593.9 2506.72   703.5 2497.56   725.8 2490.32   733.4 2488.77
   740.8 2489.12   763.3  2493.5   783.2 2499.44   803.1 2502.32   872.9 2519.38
   892.8 2521.96   922.7 2530.45   982.5 2550.54   992.4 2550.99  1022.4 2559.36
#Mann= 3 , 0 , 0
       0      .1       0   725.8    .045       0   740.8      .1       0
Bank Sta=725.8,740.8
XS Rating Curve= 0 ,0
Exp/Cntr=0.3,0.1

Type RM Length L Ch R = 1 ,38773.2 ,98.2,108.5,119.9
XS GIS Cut Line= 3
     1905623.101      215830.901     1905604.473      216007.865
      1905307.98      216240.713
#Sta/Elev= 30
       0 2549.73    29.7 2531.96    49.4 2521.64    59.3  2520.2    79.1 2515.64
    98.9 2512.59   138.4 2507.52   158.2 2505.74   177.9 2502.52   207.7 2498.87
   237.5  2493.6   287.1 2493.23     297 2492.73   316.8 2489.65   327.8 2486.97
   336.7 2484.88   342.8 2484.12   346.6 2483.65   356.5 2485.06   366.4 2488.06
   376.4 2492.88   386.3 2498.92     416 2519.96     426 2524.37   435.9 2531.02
   445.8 2541.95   455.7 2547.71   525.2 2573.79   535.1 2576.91   554.9 2585.41
#Mann= 3 , 0 , 0
       0      .1       0   327.8    .045       0   342.8      .1       0
Bank Sta=327.8,342.8
XS Rating Curve= 0 ,0
Exp/Cntr=0.3,0.1

Type RM Length L Ch R = 1 ,38664.8 ,210.3,188.5,166.8
XS GIS Cut Line= 4
      1905603.82      215936.686     1905584.468      216009.697
     1905288.025      216044.883      1905224.69       216128.45
#Sta/Elev= 30
       0 2512.14    18.9 2510.06    28.3 2508.65    37.8 2506.66    47.2 2506.56
    66.1 2501.92    85.5 2498.94   115.3 2495.29   135.2 2494.52   194.9 2493.26
   204.9 2492.43   214.8 2488.73   224.8 2483.34   231.3 2481.31   234.8 2480.21
   244.7 2481.52   246.3 2482.33   264.6 2491.83   274.6 2494.11   284.5 2494.86
   294.4 2496.55   314.4 2501.99   344.2 2511.38   364.1 2519.72   374.1 2522.47
   393.1 2530.19   412.2  2534.8   431.2 2542.24   469.4 2554.26   478.9 2558.62
#Mann= 3 , 0 , 0
       0      .1       0   231.3    .045       0   246.3      .1       0
Bank Sta=231.3,246.3
XS Rating Curve= 0 ,0
Exp/Cntr=0.3,0.1

Type RM Length L Ch R = 1 ,38476.2 ,301.5,309.6,316
XS GIS Cut Line= 3
     1905652.152      215344.296     1905258.663      216038.058
     1905107.821      216251.938
#Sta/Elev= 30
       0 2637.27    69.8 2616.83    89.7 2614.76   149.6 2600.15   179.5 2595.59
   199.4 2595.81   229.3 2591.75   299.1 2563.97     329 2545.34   348.9  2541.6
   378.8 2541.31   408.8 2531.92   438.7 2519.47   498.5 2489.61   518.4 2484.48
   548.3 2470.27   568.3 2463.87   586.1    2465   601.1 2466.14   618.1  2465.9
   628.1 2467.84   707.9  2499.3   767.7  2514.1   826.7 2539.87     846 2544.85
   865.4 2554.68   923.6 2571.46   981.8  2583.5  1001.1 2591.97  1059.3 2610.05
#Mann= 3 , 0 , 0
       0      .1       0   586.1    .045       0   601.1      .1       0
Bank Sta=586.1,601.1
XS Rating Curve= 0 ,0
Exp/Cntr=0.3,0.1

Type RM Length L Ch R = 1 ,38166.3 ,311.8,299.1,291.1
XS GIS Cut Line= 3
     1905579.927      215284.093     1905161.235      215643.714
      1904750.84      216052.847
#Sta/Elev= 30
       0 2665.42    39.4 2647.64    59.1 2641.83   147.8 2595.39   177.4 2577.99
   216.8 2564.82   256.2 2559.24   295.7 2540.76   354.8 2519.61   364.7 2515.11
   384.4  2501.8     414 2489.31   544.4 2450.84   551.9 2449.48   559.4 2449.61
   571.9 2451.19   601.9  2461.8   691.8 2483.36   731.8    2497   751.8 2500.36
   791.7 2518.52   821.7 2538.07   841.7 2540.17   881.6    2551   931.6 2573.57
   961.6 2584.33  1001.5  2593.5  1021.5 2595.52  1041.5 2601.35  1131.4 2640.99
#Mann= 3 , 0 , 0
       0      .1       0   544.4    .045       0   559.4      .1       0
Bank Sta=544.4,559.4
XS Rating Curve= 0 ,0
Exp/Cntr=0.3,0.1

Type RM Length L Ch R = 1 ,37867.1 ,295.5,299.4,302.4
XS GIS Cut Line= 3
     1905085.127      214968.335     1904922.328      215483.699
     1904679.815      216006.844
#Sta/Elev= 30
       0 2607.03      50 2614.63   150.1 2610.19   160.1 2607.37   200.2 2593.38
   250.2 2565.18   270.2 2558.11   350.3  2504.7   360.3 2503.96   420.4 2469.23
   440.4 2461.06   490.4 2447.72     533 2439.92     548 2437.84   550.4 2437.72
   649.8 2457.01   659.8 2457.01   689.6 2465.33   749.2 2488.61   759.2 2489.28
   858.6 2536.55   868.5 2537.21   898.4 2549.63   928.2 2555.15     958  2566.9
     968 2566.78  1017.7 2579.48  1057.4 2594.55  1067.4 2594.61  1117.1 2620.76
#Mann= 3 , 0 , 0
       0      .1       0     533    .045       0     548      .1       0
Bank Sta=533,548
XS Rating Curve= 0 ,0
Exp/Cntr=0.3,0.1

Type RM Length L Ch R = 1 ,37567.1 ,289,295.9,296.6
XS GIS Cut Line= 3
     1904901.116      214912.494     1904636.092      215418.435
     1904320.829      215858.385
#Sta/Elev= 30
       0 2575.21     9.8 2574.72    59.1 2584.56    78.8 2586.32    88.6 2584.88
   177.2  2545.6   216.6 2522.21   226.5 2520.28     256 2507.19   275.7 2502.03
     325 2483.27   344.7 2478.64   423.4 2452.55   554.6 2425.34   561.3 2423.56
   569.6 2423.64   610.5 2436.45   649.9 2453.16   669.6 2457.39   758.1 2501.14
   777.8 2506.72   876.2 2559.71   895.9 2566.03   935.3  2584.8   964.8  2590.6
   994.3 2605.43    1014 2611.82  1063.2 2638.48    1073 2640.87  1112.4 2639.94
#Mann= 3 , 0 , 0
       0      .1       0   554.6    .045       0   569.6      .1       0
Bank Sta=554.6,569.6
XS Rating Curve= 0 ,0
Exp/Cntr=0.3,0.1

Type RM Length L Ch R = 1 ,37271   ,301.8,296.4,291.7
XS GIS Cut Line= 3
     1904803.021      214830.251     1904419.655      215213.643
      1904101.22      215683.558
#Sta/Elev= 30
       0 2529.28    88.7 2524.46   118.3 2518.32   128.2 2513.04     138  2510.5
   226.7 2493.44   246.4 2484.51   315.4 2467.96   364.7 2449.94   453.5 2426.06
   473.2 2418.22   534.7 2404.86   549.7 2403.26   552.1 2403.07   562.1 2405.07
     592  2424.1   631.8 2446.36   651.7 2452.62   741.4 2503.64   761.3  2509.1
   791.2 2528.17     821 2541.62   850.9 2551.68   880.8 2552.45   990.3  2572.8
  1000.3 2578.41  1010.2 2587.11  1030.2 2608.56  1040.1 2615.84  1109.8 2631.39
#Mann= 3 , 0 , 0
       0      .1       0   534.7    .045       0   549.7      .1       0
Bank Sta=534.7,549.7
XS Rating Curve= 0 ,0
Exp/Cntr=0.3,0.1

Type RM Length L Ch R = 1 ,36974.5 ,275,282.1,288.9
XS GIS Cut Line= 3
     1904442.583      214626.719     1904155.185      215088.646
     1903947.394      215610.498
#Sta/Elev= 30
       0 2580.79    29.7 2578.47    49.5 2571.95    79.1  2554.5   108.8 2529.07
   128.6 2518.47     178 2484.62   217.6 2465.24   237.4 2460.75   286.8 2439.79
   385.8 2410.43   484.7 2400.47   534.2 2388.61     544 2387.73   549.2 2387.92
   563.7 2392.33   603.2  2418.5     613 2418.87   652.4 2451.56   672.1 2458.87
   731.3 2511.17     751 2524.12   760.8 2526.08   859.4 2566.09   869.2  2566.6
   957.9 2597.42   967.8  2597.2  1007.2 2609.45  1056.5 2628.58  1105.7 2632.91
#Mann= 3 , 0 , 0
       0      .1       0   534.2    .045       0   549.2      .1       0
Bank Sta=534.2,549.2
XS Rating Curve= 0 ,0
Exp/Cntr=0.3,0.1

Type RM Length L Ch R = 1 ,36692.3 ,324.7,306.7,295.5
XS GIS Cut Line= 3
     1904359.442      214567.794     1903942.819      214918.315
     1903628.701      215418.414
#Sta/Elev= 30
       0 2573.21    39.6  2567.2    59.4 2557.73    79.2 2545.21      99    2540
   217.8 2486.45   247.5 2478.44   356.4 2433.63   376.2 2429.02   425.7 2408.79
   475.2  2391.1   504.9 2375.14   524.7 2370.17   526.1 2370.17   541.1 2371.72
   583.8 2382.59     633 2398.44   642.9 2398.44   731.5 2428.14   751.2 2430.76
   810.2 2452.92   820.1 2453.53   849.6 2467.02   869.3 2470.96   967.7  2517.7
   987.4 2521.88  1036.6 2545.12  1085.8 2559.65  1105.5 2561.29    1135 2569.14
#Mann= 3 , 0 , 0
       0      .1       0   526.1    .045       0   541.1      .1       0
Bank Sta=526.1,541.1
XS Rating Curve= 0 ,0
Exp/Cntr=0.3,0.1

Type RM Length L Ch R = 1 ,36385.6 ,294.2,300.1,305.2
XS GIS Cut Line= 3
     1903732.337      214298.543      1903679.22      214837.847
       1903552.4      215392.352
#Sta/Elev= 30
       0 2567.29    29.6 2560.57    49.3    2559   137.9 2538.79   206.9 2502.62
   226.6 2499.12   256.2 2486.62   315.3 2456.31   325.2 2456.09     404  2414.5
   413.8 2413.83   423.7 2409.46   492.6 2373.28   532.1 2358.93   534.4 2358.93
   549.4  2360.1   611.8 2371.55   691.6 2398.51   701.6 2399.09   761.5 2423.54
   771.4 2423.68   801.4 2436.91   811.4 2437.59   891.2 2474.24   911.2  2478.7
     991 2512.26  1010.9 2515.77  1090.8 2549.06  1100.8 2548.89  1110.7 2552.89
#Mann= 3 , 0 , 0
       0      .1       0   534.4    .045       0   549.4      .1       0
Bank Sta=534.4,549.4
XS Rating Curve= 0 ,0
Exp/Cntr=0.3,0.1

Type RM Length L Ch R = 1 ,36085.6 ,296.9,299.7,300.2
XS GIS Cut Line= 3
     1903585.649      214276.398     1903391.577      214791.576
     1903153.039      215282.255
#Sta/Elev= 30
       0 2638.91    19.7 2629.82    39.3 2616.89    49.2 2615.34   137.6 2551.24
   157.3 2543.15   216.3 2495.67   235.9 2482.01   255.6 2475.45   294.9 2452.48
   344.1 2427.76   363.7 2422.88   442.4 2387.28     462 2382.63   511.2 2360.92
   530.9    2350   540.7 2347.75     543 2347.87     558 2348.26     610  2353.5
   649.7 2370.03   669.6 2373.83   689.4 2380.72   838.2 2438.34   887.8 2450.66
   977.1  2492.3     987 2496.36   996.9 2497.08  1086.2 2547.59  1096.1  2548.1
#Mann= 3 , 0 , 0
       0      .1       0     543    .045       0     558      .1       0
Bank Sta=543,558
XS Rating Curve= 0 ,0
Exp/Cntr=0.3,0.1

Type RM Length L Ch R = 1 ,35785.6 ,310.9,299.9,293.4
XS GIS Cut Line= 3
     1903379.866      214171.981     1903125.928      214655.194
     1902878.668      215142.345
#Sta/Elev= 30
       0 2642.35    49.6 2604.57    69.5 2593.98    99.2 2572.55   158.8 2526.17
   168.7 2524.61     258 2449.92   277.9 2442.11   337.4 2404.42   367.2 2389.21
   387.1 2383.74   406.9 2372.34   446.6 2357.28   538.4 2337.04   545.9 2335.87
   553.4 2337.17   575.7 2345.52   635.3 2350.07   684.9 2366.96   704.8 2371.26
   774.3 2413.14   794.2 2423.25   814.1  2428.9   883.6 2465.84   992.8 2533.86
  1002.8 2535.97  1012.7 2542.63  1022.6 2544.82  1032.6 2550.48  1092.2 2592.45
#Mann= 3 , 0 , 0
       0      .1       0   538.4    .045       0   553.4      .1       0
Bank Sta=538.4,553.4
XS Rating Curve= 0 ,0
Exp/Cntr=0.3,0.1

Type RM Length L Ch R = 1 ,35485.6 ,144.1,148.8,149.5
XS GIS Cut Line= 3
     1902848.923      214001.343     1902848.943      214546.148
      1902750.12      215090.015
#Sta/Elev= 30
       0 2514.72     9.9 2509.37    19.8 2509.37     109 2470.59   118.9 2470.18
   198.1 2438.96   217.9 2434.24   297.2 2400.46     317  2396.5   396.2 2369.37
     416    2366   537.3 2322.88   544.8 2321.94   552.3 2322.55   623.8 2328.82
   643.5 2333.55     683 2351.09   692.9  2351.2   781.7 2397.18   801.4 2402.55
   870.6 2444.74   890.3 2450.05   929.8 2471.38   979.1 2503.47     989 2504.55
  1058.1 2565.14    1068 2566.03  1077.8 2573.68  1087.7 2575.08  1097.6 2581.98
#Mann= 3 , 0 , 0
       0      .1       0   537.3    .045       0   552.3      .1       0
Bank Sta=537.3,552.3
XS Rating Curve= 0 ,0
Exp/Cntr=0.3,0.1

Type RM Length L Ch R = 1 ,35336.8 ,148.1,151.1,154.8
XS GIS Cut Line= 2
     1902762.282      214246.182     1902601.873      214999.263
#Sta/Elev= 30
       0 2412.81      50 2389.87      70 2385.68      80 2381.84     140 2363.85
     150 2361.22     160 2360.65     250 2331.72     260 2331.14     270 2328.06
     290 2319.47     300 2316.58     310 2317.45     340 2326.62     360 2329.58
     380 2336.17     410 2347.54     440 2360.96     460 2365.58     500  2382.5
     540 2405.26     550 2406.95     640  2455.7     650 2455.73     660 2461.02
     700  2486.4     730 2508.54     740 2510.05     750 2516.25     770 2532.65
#Mann= 3 , 0 , 0
       0      .1       0     290    .045       0     310      .1       0
Bank Sta=290,310
XS Rating Curve= 0 ,0
Exp/Cntr=0.3,0.1

Type RM Length L Ch R = 1 ,35185.6 ,144.8,148.9,152.3
XS GIS Cut Line= 3
     1902742.651      213986.174     1902553.157       214521.36
      1902354.33      215025.705
#Sta/Elev= 30
       0 2568.06    19.9 2549.04    29.9 2543.27    39.8 2541.67    79.7 2511.72
   109.6 2496.12   129.5 2482.83   149.4 2475.43   229.1 2418.18     239 2417.34
   268.9 2404.96   328.7 2372.31   428.3  2339.1   547.8 2313.39   575.2 2304.89
   577.6 2304.42   587.5 2305.48   626.9 2323.96   646.6 2329.21   725.4 2371.32
   745.2 2377.61   794.4 2407.52   873.3    2432   932.4 2467.38   942.3 2469.38
   971.9 2485.04  1021.2 2516.05  1040.9 2526.04  1060.6 2532.38  1109.9 2558.38
#Mann= 3 , 0 , 0
       0      .1       0   575.2    .045       0   587.5      .1       0
Bank Sta=575.2,587.5
XS Rating Curve= 0 ,0
Exp/Cntr=0.3,0.1

Type RM Length L Ch R = 1 ,35036.5 ,157.8,152,146.3
XS GIS Cut Line= 2
     1902573.168       214190.46     1902270.922       214717.28
#Sta/Elev= 30
       0 2407.02      10 2403.95    19.9 2402.56    29.9  2400.1    39.8 2395.27
    59.7 2380.44    69.7 2375.05   109.5 2357.76   119.5 2354.58   129.4 2353.41
   209.1 2322.25     229 2313.27   248.9 2309.22   279.2 2297.62   288.8 2295.28
   294.2 2295.54   298.7 2295.76   328.6 2301.98   348.5 2304.03   358.4 2306.88
   368.4 2310.92   388.3 2321.09   448.1 2349.87     458 2351.78     468 2354.84
   507.8 2375.38   547.6 2400.18   557.6 2404.87   567.5 2405.95   607.4 2430.62
#Mann= 3 , 0 , 0
       0      .1       0   279.2    .045       0   294.2      .1       0
Bank Sta=279.2,294.2
XS Rating Curve= 0 ,0
Exp/Cntr=0.3,0.1

Type RM Length L Ch R = 1 ,34884.4 ,306.9,302.4,296.7
XS GIS Cut Line= 3
     1902434.058      213863.403     1902290.936      214389.665
     1902127.399      214914.393
#Sta/Elev= 30
       0 2526.52    19.8 2511.01    49.6 2492.58    59.5 2491.93   138.8  2451.4
   158.6 2445.84     238 2404.74   287.6  2387.8   337.1 2364.62     357 2359.45
   436.3 2320.95   456.1 2315.99   515.6 2287.54   521.4 2287.66   536.4 2291.02
   545.4 2291.53   635.3  2316.5   655.3 2319.35   695.3 2334.24   735.2 2353.82
   745.2 2354.55   835.2 2410.21   855.2  2417.2   895.1    2445   935.1 2479.73
   945.1 2480.46    1025 2536.11    1035 2542.11    1055 2547.75    1095 2573.26
#Mann= 3 , 0 , 0
       0      .1       0   521.4    .045       0   536.4      .1       0
Bank Sta=521.4,536.4
XS Rating Curve= 0 ,0
Exp/Cntr=0.3,0.1

Type RM Length L Ch R = 1 ,34581.9 ,291.4,300,303.8
XS GIS Cut Line= 3
     1902032.272      213810.114     1901994.486      214359.588
     1901982.653      214904.617
#Sta/Elev= 30
       0 2459.43    68.8  2449.8   108.2 2438.21   186.9 2408.56   206.5 2405.52
   245.9 2392.95   275.4 2378.78   295.1 2373.39   344.2 2338.42   373.7 2322.37
   442.6 2304.28   472.1  2293.8   481.9  2293.6   543.3 2268.18   550.8 2267.05
   558.3 2268.89   570.6 2273.68   590.4 2277.43   659.8 2305.99   679.6 2310.45
   758.9 2351.49   778.8 2357.05   818.4 2380.64   848.1 2400.32     868 2407.33
   947.2  2461.6   967.1  2467.4  1036.5 2507.85  1056.3 2513.08  1095.9 2534.06
#Mann= 3 , 0 , 0
       0      .1       0   543.3    .045       0   558.3      .1       0
Bank Sta=543.3,558.3
XS Rating Curve= 0 ,0
Exp/Cntr=0.3,0.1
